--- LONGRN.prj (project) ---

Proj Title=LONGRN
Current Plan=p01
Default Exp/Contr=0,0
English Units
Geom File=g01
Flow File=f01
Plan File=p01
BEGIN DESCRIPTION:
Stream Name: Long Run
Flood Zone: Approximate
Pendleton County, West Virginia
HEC-RAS Version: 5.0.7
Hydrology Method:
Regression equation
END DESCRIPTION:
DSS Export Rating Curves= 0
DSS Export Rating Curve Sorted= 0
DSS Export Volume Flow Curves= 0
DXF OffsetX= 0
DXF OffsetY= 0
DXF ScaleX= 0
DXF ScaleY= 0

--- LONGRN.p01 (plan) ---

Plan Title=Floodplain
Program Version=5.07
Short Identifier=Floodplain
Geom File=g01
Flow File=f01
Subcritical Flow
K Sum by GR= 0
Std Step Tol= 0.01
Critical Tol= 0.01
Num of Std Step Trials= 20
Max Error Tol= 0.3
Flow Tol Ratio= 0.001
Split Flow NTrial= 30
Split Flow Tol= 0.02
Split Flow Ratio= 0.02
Log Output Level= 0
Friction Slope Method= 1
Unsteady Friction Slope Method= 2
Unsteady Bridges Friction Slope Method= 1
Parabolic Critical Depth
Global Vel Dist= 0 , 0 , 0
Global Log Level= 0
CheckData=True
Encroach Param=-1 ,0,0, 0
Mapping Interval=1HOUR
Computation Time Step Use Courant=        0
Computation Time Step Use Time Series=    0
Computation Time Step Count To Double=0
Computation Time Step Max Doubling=0
Computation Time Step Max Halving=0
Computation Time Step Residence Courant=0
Run HTab= 0
Run UNet= 0
Run Sediment= 0
Run PostProcess= 0
Run WQNet= 0
Run RASMapper= 0
UNET Theta= 0
UNET Theta Warmup= 0
UNET ZTol= 0
UNET ZSATol= 0
UNET MxIter= 0
UNET Max Iter WO Improvement= 0
UNET MaxInSteps= 0
UNET DtIC= 0
UNET DtMin= 0
UNET MaxCRTS= 0
UNET WFStab= 0
UNET SFStab= 0
UNET WFX= 1
UNET SFX= 1
UNET 1D Methodology=Finite Difference
UNET DSS MLevel= 1
UNET Pardiso=0
UNET DZMax Abort= 0
UNET Use Existing IB Tables= 0
UNET Froude Reduction=False
UNET Froude Limit= 0
UNET Froude Power= 0
UNET D1 Cores= 0
UNET D2 Coriolis=0
UNET D2 Cores= 0
UNET D2 Theta= 1
UNET D2 Theta Warmup= 1
UNET D2 Z Tol= 0.01
UNET D2 Volume Tol= 0.01
UNET D2 Max Iterations= 20
UNET D2 Equation= 0
UNET D2 RampUpFraction=0.1
UNET D2 TimeSlices= 1
UNET D2 BCVolumeCheck=0
UNET D1D2 MaxIter= 0
UNET D1D2 ZTol=0.01
UNET D1D2 QTol=0.1
UNET D1D2 MinQTol=1
Write IC File= 0
Write IC File at Fixed DateTime=0
Write IC File at Sim End=0
Echo Input=False
Echo Parameters=False
Echo Output=False
Write Detailed= 0
HDF Write Warmup=0
HDF Write Time Slices=0
HDF Flush=0
HDF Face Node Velocities=0
HDF Compression= 1
HDF Chunk Size= 1
HDF Spatial Parts= 1
HDF Use Max Rows=0
HDF Fixed Rows= 1
Calibration Method= 0
Calibration Iterations= 20
Calibration Max Change=0.05
Calibration Tolerance=0.2
Calibration Maximum=1.5
Calibration Minimum=0.5
Calibration Optimization Method= 1
WQ AD Non Conservative
WQ ULTIMATE=-1
WQ Max Comp Step=1HOUR
WQ Output Interval=15MIN
WQ Output Selected Increments= 0
WQ Output face flow=0
WQ Output face velocity=0
WQ Output face area=0
WQ Output face dispersion=0
WQ Output cell volume=0
WQ Output cell surface area=0
WQ Output cell continuity=0
WQ Output cumulative cell continuity=0
WQ Output face conc=0
WQ Output face dconc_dx=0
WQ Output face courant=0
WQ Output face peclet=0
WQ Output face adv mass=0
WQ Output face disp mass=0
WQ Output cell mass=0
WQ Output cell source sink temp=0
WQ Output nsm pathways=0
WQ Output nsm derived pathways=0
WQ Output MaxMinRange=-1
WQ Daily Max Min Mean=-1
WQ Daily Range=0
WQ Daily Time=0
WQ Create Restart=0
WQ Fixed Restart=0
WQ System Summary=0
WQ Write To DSS=0
WQ Use Fixed Temperature=0
Sorting and Armoring Iterations= 10
XS Update Threshold= 0.02
Bed Roughness Predictor= 0
Hydraulics Update Threshold= 0.02
Energy Slope Method= 1
Volume Change Method= 1
Sediment Retention Method= 0
XS Weighting Method= 0
Number of US Weighted Cross Sections= 1
Number of DS Weighted Cross Sections= 1
Upstream XS Weight=0
Main XS Weight=1
Downstream XS Weight=0
Number of DS XS's Weighted with US Boundary= 1
Upstream Boundary Weight= 1
Weight of XSs Associated with US Boundary= 0
Number of US XS's Weighted with DS Boundary= 1
Downstream Boundary Weight= 0.5
Weight of XSs Associated with DS Boundary= 0.5
Percentile Method= 0
Sediment Output Level= 3
Mass or Volume Output= 0
Output Increment Type= 1
Profile and TS Output Increment= 1
XS Output Flag= 0
XS Output Increment= 10
Write Gradation File= 0
Read Gradation Hotstart= 0
Write HDF5 File= 1
Write Binary Output= 1
Write DSS Sediment File= 0
SV Curve= 0
Specific Gage Flag= 0

--- LONGRN.f01 (steady flow) ---

Flow Title=Flows
Program Version=5.07
Number of Profiles= 6
Profile Names=P100yr,P10yr,P25yr,P50yr,P500yr,P101yr
River Rch & RM=LONGRN,Main            ,12533
     807     376     532     665    1187     982
River Rch & RM=LONGRN,Main            ,10276
     900     418     593     742    1325    1095
River Rch & RM=LONGRN,Main            ,8887
    1005     466     661     828    1482    1223
River Rch & RM=LONGRN,Main            ,6836
    1146     531     754     944    1693    1395
River Rch & RM=LONGRN,Main            ,3986
    1278     591     839    1052    1889    1555
River Rch & RM=LONGRN,Main            ,0
    1790     823    1173    1472    2656    2179
Boundary for River Rch & Prof#=LONGRN,Main            , 1
Up Type= 0
Dn Type= 1
Dn Known WS=2293.66
Boundary for River Rch & Prof#=LONGRN,Main            , 2
Up Type= 0
Dn Type= 1
Dn Known WS=2291.96
Boundary for River Rch & Prof#=LONGRN,Main            , 3
Up Type= 0
Dn Type= 1
Dn Known WS=2292.64
Boundary for River Rch & Prof#=LONGRN,Main            , 4
Up Type= 0
Dn Type= 1
Dn Known WS=2293.15
Boundary for River Rch & Prof#=LONGRN,Main            , 5
Up Type= 0
Dn Type= 1
Dn Known WS=2294.85
Boundary for River Rch & Prof#=LONGRN,Main            , 6
Up Type= 0
Dn Type= 1
Dn Known WS=2294.21
DSS Import GetInterval= 0
DSS Import GetPeak= 0
DSS Import FillOption= 0

--- LONGRN.g01 (geometry) ---

Geom Title=Geometry
Program Version=5.07

River Reach=LONGRN          ,Main
Reach XY= 30
     2415931.719      700145.547     2416275.332      699963.416
     2416451.747      699728.882     2416698.783      699676.132
     2416867.082      699492.124     2417285.626      699390.434
     2417872.575      699030.782     2418301.435      699007.869
     2418421.946      698815.622     2418664.203      698715.461
     2418980.771      698729.014     2419918.494      697836.951
      2420012.86      697668.342     2420412.682       697559.27
     2420386.563      697295.745     2420551.176      697041.551
     2420398.495      696798.994     2420500.842      696461.634
     2420674.965      696409.486      2421278.95      695913.403
     2421271.426      695428.207     2421631.285      695239.554
     2421697.658      695053.973     2422175.269      694508.674
     2422060.567      694148.976     2422294.053       693917.95
     2422355.362      693646.601     2422857.728      693213.129
     2422877.922      692876.613       2423197.7      692365.156

Type RM Length L Ch R = 1 ,12533   ,297.1,297.1,297.1
XS GIS Cut Line= 2
2416193.84784425700491.5213236432415701.93812368 699842.26758208
#Sta/Elev= 30
       0 3305.74    86.1  3239.8   125.4 3212.14   231.6 3148.12   302.5 3109.41
   328.2 3092.09   342.9 3078.82   382.4 3050.48   392.2 3046.37   412.3 3043.45
   425.2 3030.68   442.3 3029.35   444.4 3029.35   455.5 3030.65   468.1 3035.13
     508 3057.95   522.7 3058.69   541.7 3053.76   561.5 3052.37   582.9 3055.51
   618.1 3074.64   628.1 3077.16   653.2 3077.67   707.2 3070.64   718.4 3071.09
   733.5  3078.1   747.9 3080.96   759.3 3087.71   783.7 3095.88   814.6 3109.91
#Mann= 3 , 0 , 0
       0      .1       0   425.2    .045       0   444.4      .1       0
Bank Sta=425.2,444.4
XS Rating Curve= 0 ,0
Exp/Cntr(USF)=0,0
Exp/Cntr=0.3,0.1

Type RM Length L Ch R = 1 ,12236   ,162.2,156.6,153.6
XS GIS Cut Line= 3
2416394.28198263700375.801017371     2416176.399      700006.392
     2415967.829      699656.661
#Sta/Elev= 30
       0 3258.13    22.7 3240.62    55.8 3219.57    67.5 3210.45     145 3163.21
   330.8 3058.58     377 3027.82   392.8 3019.06   403.4  3009.7   414.4 3009.02
   428.9 3006.33   439.9 3009.01   446.9 3012.65   458.9 3024.32   470.2  3031.8
   488.8 3037.99   502.4 3039.79   516.8 3037.77   535.4 3038.73     568 3032.68
   600.6 3034.89   609.9 3038.56   623.9 3047.03   636.9 3049.01   648.5 3053.54
   671.9 3058.48   692.3 3064.97     704 3066.67   791.6 3106.79   836.1 3131.49
#Mann= 3 ,-1 , 0
       0      .1       0   414.4    .045       0   439.9      .1       0
Bank Sta=414.4,439.9
XS Rating Curve= 0 ,0
Exp/Cntr=0.3,0.1

Type RM Length L Ch R = 1 ,12079   ,147.3,143.4,140.2
XS GIS Cut Line= 2
2416598.01914324700232.1346861272416014.79533302 699628.13852102
#Sta/Elev= 30
       0 3215.72    17.3 3204.59    96.5 3161.67   206.3 3107.98   300.2 3059.47
   321.4 3049.57   362.5 3033.07   373.3 3024.45   390.7 3006.66   396.5 3002.65
     402 3002.13     436 3002.87   447.3 3006.36   476.9 3007.42   503.9 3011.23
   552.2 3013.91   563.3 3019.79     580 3031.86   594.4 3035.12   603.6 3039.64
   628.4 3043.65   652.3 3049.38   696.8 3065.25   713.2 3073.51   735.7 3078.95
   747.2 3085.06   770.6 3094.27   806.6 3110.62   830.2 3123.56   839.6  3125.4
#Mann= 3 ,-1 , 0
       0      .1       0   396.5    .045       0     436      .1       0
Bank Sta=396.5,436
XS Rating Curve= 0 ,0
Exp/Cntr(USF)=0,0
Exp/Cntr=0.3,0.1

Type RM Length L Ch R = 1 ,11936   ,398.8,393.7,395.9
XS GIS Cut Line= 3
2416726.24605211700071.617051321     2416393.521       699818.58
     2416052.716      699579.416
#Sta/Elev= 30
       0 3152.83    74.8  3123.4    93.7 3113.47   220.5  3059.7   274.2 3042.52
   300.9  3031.4     337 3020.44   354.1 3017.05     377 3014.96   386.3 3009.66
   401.4 2996.29   408.4 2992.18   431.4 2990.25   442.8  2991.9     460 2994.16
   475.2    2993   485.8 2993.68   523.2 3018.63   533.8 3019.56   558.2 3025.58
   621.8 3043.55   709.8 3080.71   724.4 3088.62   738.5 3090.85   761.5 3102.93
   770.1 3109.19   787.9 3111.45   793.5 3113.89   802.6 3120.44   834.4  3133.7
#Mann= 3 ,-1 , 0
       0      .1       0   408.4    .045       0   442.8      .1       0
#XS Ineff= 2 , 0
       0                   462.9       0    2998
Permanent Ineff=
       F       F
Bank Sta=408.4,442.8
XS Rating Curve= 0 ,0
Exp/Cntr=0.3,0.1

Type RM Length L Ch R = 1 ,11542   ,464.5,478.4,479.2
XS GIS Cut Line= 3
2417026.26743509699867.3952456242416516.85018249699532.034072096
     2416443.419      699290.147
#Sta/Elev= 30
       0 3101.19   146.4 3050.38   196.4 3035.56   236.8 3021.24   277.3 3013.61
   310.7 3003.22   325.1 2996.03   334.7  2988.9   346.6 2977.96   355.2 2967.05
   358.6 2964.01   366.8 2962.29   382.5 2962.15   393.7 2963.72   401.7 2965.09
   420.9 2964.74     439 2968.82   473.8 2987.58   521.4 2998.62   559.7 3011.74
   569.3 3016.53   583.7 3018.83     598 3026.33   670.2 3057.05   774.1 3098.63
   799.2 3111.29   814.5 3114.03   828.5 3123.31     841 3126.96   862.7 3138.43
#Mann= 3 ,-1 , 0
       0      .1       0   358.6    .045       0   393.7      .1       0
Bank Sta=358.6,393.7
XS Rating Curve= 0 ,0
Exp/Cntr=0.3,0.1

Type RM Length L Ch R = 1 ,11064   ,362.7,356.8,352
XS GIS Cut Line= 2
 2417300.1535734699804.7716110422416865.67564757699091.178393962
#Sta/Elev= 30
       0 3140.82    54.8 3108.52   124.6 3071.67   161.4 3053.72   231.7  3022.5
   281.8 2998.26   325.8 2980.27   348.6 2967.63   360.6  2962.9   381.5 2948.01
   392.4 2941.58   409.6 2936.99   420.5 2932.55   430.3 2931.51   451.8 2932.31
   465.8 2930.52   475.2 2931.38   482.7 2934.13   503.1 2950.94   512.7  2957.4
   559.5 2961.05   582.9 2969.53     611  2983.5   615.7 2984.98   625.1 2985.26
   639.1 2991.33   681.3 2998.76   741.1  3003.1   762.1  3010.2   835.5 3029.59
#Mann= 3 ,-1 , 0
       0      .1       0   420.5    .045       0   451.8      .1       0
Bank Sta=420.5,451.8
XS Rating Curve= 0 ,0
Exp/Cntr=0.3,0.1

Type RM Length L Ch R = 1 ,10707   ,416.2,431.2,431.6
XS GIS Cut Line= 2
2417657.33141754699593.3130350962417073.81438913699012.982337184
#Sta/Elev= 30
       0 3061.51    77.2  3028.2   161.9 2993.25   215.7 2975.58   241.7 2965.76
   338.1 2923.17   360.8 2915.91   385.4 2911.78   398.5 2909.89   411.8 2910.19
   423.2 2911.71   430.6 2912.46   443.7 2917.17   456.1 2919.43   485.6 2934.35
   496.9 2941.37     517 2947.69   562.1  2957.7     582 2964.93   593.4 2966.05
   604.7 2970.53   621.7 2974.49   638.7  2980.2   690.9 2991.43   708.8 2996.37
   730.5 3004.66   765.2  3023.4   774.9 3026.04   803.2 3037.86     823 3044.75
#Mann= 3 ,-1 , 0
       0      .1       0   385.4    .045       0   423.2      .1       0
Bank Sta=385.4,423.2
XS Rating Curve= 0 ,0
Exp/Cntr=0.3,0.1

Type RM Length L Ch R = 1 ,10276   ,330.1,343.7,346.5
XS GIS Cut Line= 3
     2417922.566      699486.0292417736.64591052      699126.088
     2417551.932       698751.48
#Sta/Elev= 30
       0 3047.19    21.5 3034.58    58.6 3015.74   129.6 2983.02   200.1 2955.63
   282.7 2921.61   318.7 2909.59   355.5 2890.98   388.1 2887.93   408.7 2885.81
   417.6 2885.99   423.9 2887.78     431 2890.85   441.8 2892.11   469.6 2902.22
   492.6 2912.68   506.8 2920.67   520.2 2923.08   529.1 2928.95   573.7 2947.05
   591.1 2955.93   613.8 2963.76   649.5 2980.43   662.7 2984.83   685.2 2994.34
     703 3004.78   707.5 3006.59   725.3 3010.29   747.6 3023.74   822.8 3058.41
#Mann= 3 ,-1 , 0
       0      .1       0   388.1    .045       0   423.9      .1       0
Bank Sta=388.1,423.9
XS Rating Curve= 0 ,0
Exp/Cntr=0.3,0.1

Type RM Length L Ch R = 1 ,9932    ,252.9,246.1,241.7
XS GIS Cut Line= 2
2418051.80172675 699473.013693062418032.32424158698657.688886321
#Sta/Elev= 30
       0 3061.36     6.1 3056.22    34.4 3037.61    62.1 3020.87   155.5 2973.06
   218.3 2947.33   250.2 2935.74   286.2 2920.27   358.2 2897.52   386.1 2885.01
     411 2870.33   430.2 2868.49   443.8 2869.86   458.3 2874.86   478.3 2875.78
   514.3  2888.5   530.7 2892.12   550.4 2898.42   566.3 2906.05   578.3 2906.68
   590.3 2913.34   610.3 2921.24   626.3 2925.45   658.3 2936.82   694.3 2951.38
   710.3 2959.94   726.3 2962.41   738.3  2970.4   750.3  2974.8   815.6 3006.33
#Mann= 3 ,-1 , 0
       0      .1       0     411    .045       0   443.8      .1       0
Bank Sta=411,443.8
XS Rating Curve= 0 ,0
Exp/Cntr=0.3,0.1

Type RM Length L Ch R = 1 ,9686    ,289.5,287.2,288.5
XS GIS Cut Line= 3
2418446.22271742699380.534193666     2418281.188      699015.357
      2418055.25      698608.145
#Sta/Elev= 30
       0 2972.11    45.7 2969.74    64.3 2966.86   102.8 2959.19     155 2945.53
   216.9 2919.58   256.4 2907.29   295.9  2892.4   354.6 2861.24   363.6 2859.72
   381.8 2860.33   400.7 2858.36   408.2 2860.04   419.6 2863.28   467.6 2859.58
   497.3 2860.49   511.1 2864.72   533.9 2867.01     566 2880.37   579.7 2888.43
   593.4 2891.22   611.7 2902.07   702.6 2938.06   726.1 2948.97   739.8 2957.73
     753 2960.57   761.8 2967.53   785.3 2981.07   850.1 3014.38   866.4 3024.56
#Mann= 3 ,-1 , 0
       0      .1       0   381.8    .045       0   408.2      .1       0
#XS Ineff= 2 , 0
                          419.42         2868.81
Permanent Ineff=
       F       F
Bank Sta=381.8,408.2
XS Rating Curve= 0 ,0
Exp/Cntr=0.3,0.1

Type RM Length L Ch R = 1 ,9398    ,213.7,215.5,216.2
XS GIS Cut Line= 2
2418651.28652991699295.7808428662418301.35224378698477.669635102
#Sta/Elev= 30
       0 2936.82    66.2 2916.81   109.7 2911.35   177.8 2899.54   253.3  2883.9
   288.1 2882.16   367.5 2870.21   405.6 2862.19   438.7 2861.25   458.2 2853.69
   479.5 2849.53   489.6 2848.93     510 2852.38   519.1 2847.43   530.3 2844.96
   540.4 2847.43   540.4 2847.44   549.1 2850.95   564.8 2866.04   581.1 2874.92
   611.6 2886.73   628.8 2888.55   637.9 2892.33   675.3 2901.13   723.2 2919.79
   733.7 2921.81   765.9 2938.76   779.7 2940.82   801.5 2954.29   889.8 2998.85
#Mann= 3 ,-1 , 0
       0      .1       0   519.1    .045       0   540.4      .1       0
#XS Ineff= 2 , 0
          508.13 2859.18
Permanent Ineff=
       F       F
Bank Sta=519.1,540.4
XS Rating Curve= 0 ,0
Exp/Cntr(USF)=0,0
Exp/Cntr=0.3,0.1

Type RM Length L Ch R = 1 ,9183    ,303.9,295.8,293.9
XS GIS Cut Line= 2
 2418790.6777307699263.5475833292418520.78759397698315.841930741
#Sta/Elev= 30
       0 2969.81   108.8 2921.45   237.7 2876.58   358.4  2859.4   394.1  2852.2
   424.9 2842.63   449.9 2842.49     479 2839.78   495.8 2835.48   528.1 2832.92
   537.8  2833.5   547.7 2828.25   554.7 2827.13   566.3 2828.05   603.7 2827.51
   616.2  2828.7   624.5 2834.07   654.4 2860.47   674.4 2871.92   686.9 2872.15
   770.1 2896.03   803.4 2906.68   811.7 2911.21   828.3 2913.31   846.8 2924.45
   864.8 2931.15   932.3 2962.41   957.3 2972.41   973.9 2982.38   985.4 2983.06
#Mann= 3 ,-1 , 0
       0      .1       0   547.7    .045       0   566.3      .1       0
Bank Sta=547.7,566.3
XS Rating Curve= 0 ,0
Exp/Cntr=0.3,0.1

Type RM Length L Ch R = 1 ,8887    ,341.4,331.8,322.1
XS GIS Cut Line= 2
2419049.89413905  699229.23456772418799.78391394698287.787034346
#Sta/Elev= 30
       0 3027.71    60.4 2999.05    93.5 2981.58   159.7 2943.19   229.9 2908.73
   295.5 2879.49   341.8 2861.95   429.6 2832.25   442.7 2822.87   461.8 2804.29
   466.7 2801.95   504.8 2801.42   514.6 2799.91   573.5 2802.93   604.3 2810.97
   631.5 2809.84   668.3 2810.93   710.2 2809.99     737 2819.35   772.2  2835.1
   784.6 2835.86   799.1 2841.96   830.2 2851.83   859.1  2859.7   875.7 2865.64
   893.9 2868.01   929.9 2880.61   946.1 2881.44   954.3 2886.44   974.1 2894.17
#Mann= 3 ,-1 , 0
       0      .1       0   466.7    .045       0   504.8      .1       0
Bank Sta=466.7,504.8
XS Rating Curve= 0 ,0
Exp/Cntr=0.3,0.1

Type RM Length L Ch R = 1 ,8555    ,171.7,171.2,166.6
XS GIS Cut Line= 3
2419462.57996565698842.0748791942419162.26518989698541.854103038
     2418849.117      698271.201
#Sta/Elev= 30
       0 2978.83    39.4 2962.97    64.4 2950.54   106.8 2926.39   185.6 2885.04
   191.6 2879.83   220.3 2863.88   310.8 2816.92   372.3 2794.32   377.9 2790.85
   389.2 2778.82   392.5 2777.07   412.7 2776.76   423.6 2775.97   437.7  2777.3
   450.4  2782.3   487.5 2779.04   525.7 2783.53   550.9 2788.53   565.4 2788.98
   576.7 2792.01   612.7 2794.41   624.9 2798.76     680 2827.59     693 2828.62
   704.4 2833.86   751.8 2848.72   772.9 2859.52   815.2 2865.96   838.5 2878.33
#Mann= 3 ,-1 , 0
       0      .1       0   412.7    .045       0   437.7      .1       0
#XS Ineff= 2 , 0
                          452.75         2788.86
Permanent Ineff=
       F       F
Bank Sta=412.7,437.7
XS Rating Curve= 0 ,0
Exp/Cntr=0.3,0.1

Type RM Length L Ch R = 1 ,8384    ,165.4,170.6,173.8
XS GIS Cut Line= 3
2419607.60770865698685.4937741822419285.68670865698430.634774182
2418954.10570864698179.269774182
#Sta/Elev= 30
       0 2945.77    31.7  2942.3    59.4  2935.6    62.3  2934.1    68.6  2924.7
    72.5 2921.17    87.8 2915.76   124.9 2899.08   261.6 2831.22   352.2 2791.51
   378.3 2776.43   395.4 2763.67   415.4 2761.77   432.5 2763.44   456.5 2771.37
   469.5 2773.13   484.6 2772.34   524.7 2765.35   544.8 2768.36   558.1 2774.41
   589.5 2798.18   603.8 2805.63   635.2 2810.88   672.3 2821.23   708.1 2833.52
   750.6 2844.04   789.4  2857.6   803.7 2859.44   812.2    2863   826.7 2865.93
#Mann= 3 ,-1 , 0
       0      .1       0   395.4    .045       0   432.5      .1       0
#XS Ineff= 2 , 0
                          473.31         2783.89
Permanent Ineff=
       F       F
Bank Sta=395.4,432.5
XS Rating Curve= 0 ,0
Exp/Cntr=0.3,0.1

Type RM Length L Ch R = 1 ,8214    ,330.7,327.8,319.4
XS GIS Cut Line= 2
2419629.96972009698658.0312684582419162.74272009697971.090268458
#Sta/Elev= 30
       0 2925.15    18.3 2918.89    42.5 2915.52      57 2908.91    90.9  2896.9
   162.9 2861.37   289.2 2805.37   298.3 2799.86     340 2767.15   366.6 2752.63
   376.3 2750.56   425.4 2746.24     444  2745.4   453.8 2747.21   475.2 2753.69
   516.6 2749.62   537.2 2753.85   560.1 2765.43   574.7 2765.81   583.3 2769.43
     594 2771.56   610.3  2780.6   645.8 2796.79   666.5 2803.76   718.6 2817.42
   738.3 2825.87   761.8 2827.73   773.3 2833.34   811.7 2846.06   830.8  2854.9
#Mann= 3 ,-1 , 0
       0      .1       0   425.4    .045       0   453.8      .1       0
#XS Ineff= 2 , 0
                          476.58         2758.26
Permanent Ineff=
       F       F
Bank Sta=425.4,453.8
XS Rating Curve= 0 ,0
Exp/Cntr=0.3,0.1

Type RM Length L Ch R = 1 ,7886    ,290.7,300,303.5
XS GIS Cut Line= 3
     2419973.389      698343.998     2419642.536      698110.689
     2419290.676       697854.65
#Sta/Elev= 30
       0 2898.04    22.8 2888.62    42.4 2876.56   101.1 2847.86     195 2806.22
   277.3 2782.72   336.1 2772.19   345.9 2765.48   389.9 2722.03   393.1 2720.16
   404.5 2719.34   424.6 2720.97   439.2 2723.67     459 2730.16   493.6 2729.68
   499.7 2730.79   513.4 2737.24   523.3 2740.06   547.3 2741.42   572.8 2746.23
   602.5 2757.37     656 2782.72   710.4 2804.16   726.1 2807.61   745.9 2815.86
   765.3 2817.99   775.6 2823.57   805.6 2832.17     826 2840.85     840 2843.45
#Mann= 3 ,-1 , 0
       0      .1       0   393.1    .045       0   424.6      .1       0
Bank Sta=393.1,424.6
XS Rating Curve= 0 ,0
Exp/Cntr=0.3,0.1

Type RM Length L Ch R = 1 ,7586    ,302.6,300,292.6
XS GIS Cut Line= 3
2420045.88028258698248.137523754     2419808.455      697881.354
     2419590.073      697535.637
#Sta/Elev= 30
       0 2885.63    58.1 2851.04   115.8 2821.32   182.5 2794.04     235 2776.06
   277.8  2759.1   292.4 2750.07   320.7 2728.73   349.3 2714.15   387.4 2707.71
     411 2707.89   416.8 2704.09   425.3 2702.41   455.1 2703.61   458.8 2705.79
   468.2 2717.43     473 2719.61     524  2732.4   558.1 2738.03   600.7 2756.01
   663.2 2769.71   685.9 2777.83   700.1 2784.89   723.7 2786.38   732.2 2792.67
     756 2803.01   764.7 2802.84   799.6 2814.45   818.3 2817.49   845.8 2825.35
#Mann= 3 ,-1 , 0
       0      .1       0   416.8    .045       0   455.1      .1       0
Bank Sta=416.8,455.1
XS Rating Curve= 0 ,0
Exp/Cntr=0.3,0.1

Type RM Length L Ch R = 1 ,7286    ,160.3,166.3,165.5
XS GIS Cut Line= 3
2420350.12767601697977.636339824      2419998.62      697683.616
     2419672.528      697447.712
#Sta/Elev= 30
       0 2846.27      10 2841.86    32.7 2826.17    61.8  2808.2   129.6  2772.5
   153.9 2756.17     213 2724.12     235 2714.71   284.8 2706.19   384.9 2704.65
   416.1 2691.81   442.5  2686.5   447.3 2684.72   458.1 2684.06     463 2684.32
     468 2686.31   478.7 2695.87   510.3 2715.85   527.4 2728.76   561.9 2748.49
   576.1 2751.09   587.6 2756.25     622  2767.5   650.6  2771.3   660.5  2775.6
   677.9 2778.33   691.5 2783.66   750.9 2799.76   802.4 2817.33   860.7 2833.53
#Mann= 3 ,-1 , 0
       0      .1       0   442.5    .045       0     468      .1       0
Bank Sta=442.5,468
XS Rating Curve= 0 ,0
Exp/Cntr=0.3,0.1

Type RM Length L Ch R = 1 ,7119    ,293.6,283.7,284.1
XS GIS Cut Line= 2
2420365.85334461697941.2495891962419955.73249176697346.485581815
#Sta/Elev= 30
       0 2836.56    26.6 2818.92    93.1 2781.96   124.3 2761.28   134.1 2756.76
   170.7 2732.86   223.9 2701.82   254.1 2693.36   284.7 2689.18   311.6 2687.83
   328.4 2684.27   357.6 2684.25   369.2 2679.09   383.5 2677.92   406.5 2679.56
   429.5 2682.63   443.9 2681.11   449.7 2682.37   455.4 2687.31   464.4 2698.67
   470.5 2703.72   487.1 2714.49   508.2 2731.36   517.9 2735.62   526.9 2737.43
   570.5 2740.59     605 2744.95   645.2    2754   692.8 2762.34   722.5  2770.9
#Mann= 3 ,-1 , 0
       0      .1       0   369.2    .045       0   406.5      .1       0
#XS Ineff= 2 , 0
                          430.58         2690.48
Permanent Ineff=
       F       F
Bank Sta=369.2,406.5
XS Rating Curve= 0 ,0
Exp/Cntr(USF)=0,0
Exp/Cntr=0.3,0.1

Type RM Length L Ch R = 1 ,6836    ,365.4,349.2,351.3
XS GIS Cut Line= 3
     2420714.221      697801.546     2420414.906      697556.668
     2419989.757      697227.074
#Sta/Elev= 30
       0 2791.23    35.5 2781.03    45.8 2782.03    64.1 2789.51   130.5 2788.55
   164.7 2784.28   200.5 2774.09     246 2757.04   262.9 2748.27   302.8 2703.31
   336.9 2675.41   359.7 2660.15   370.6 2658.43   396.7 2660.42   407.2 2669.07
   412.2 2670.28   448.4 2670.77     468 2673.95   493.2 2687.52   502.1 2690.26
   536.4 2689.66   590.5  2684.5   619.7 2688.41   653.2 2700.41     721 2713.08
   761.5 2726.86   812.1 2731.42   822.2 2736.73   879.3 2752.72   924.7 2774.95
#Mann= 3 ,-1 , 0
       0      .1       0   359.7    .045       0   396.7      .1       0
Bank Sta=359.7,396.7
XS Rating Curve= 0 ,0
Exp/Cntr=0.3,0.1

Type RM Length L Ch R = 1 ,6487    ,304.6,291.3,284.4
XS GIS Cut Line= 2
     2420846.353      697371.588       2420029.4      697113.073
#Sta/Elev= 30
       0 2815.66      64 2793.65   137.3 2763.76   188.3 2740.71   213.6 2727.63
   274.3 2687.42   309.4 2668.53     331 2663.01   381.4 2659.33   398.2  2652.8
   410.7 2651.66   419.1 2643.09   423.3 2641.48   439.8 2640.55   444.12638.768
   452.7 2637.18   477.9 2637.51   482.1 2639.18   515.6 2670.27   528.2 2678.22
     545 2680.53   603.7 2681.03   670.9 2690.55   704.6 2697.51   750.6 2708.52
   788.3  2723.8   805.1  2724.3   809.3 2726.26   817.7 2733.73   856.9 2756.76
#Mann= 3 ,-1 , 0
       0      .1       0   444.1    .045       0   482.1      .1       0
Bank Sta=444.1,482.1
XS Rating Curve= 0 ,0
Exp/Cntr=0.3,0.1

Type RM Length L Ch R = 1 ,6195    ,145.4,133.4,121.3
XS GIS Cut Line= 2
2420903.34848835696973.5667110652420031.61974917697053.460383698
#Sta/Elev= 30
       0 2765.32    80.9 2740.25   141.2 2724.51   161.3 2720.67   189.4 2712.23
   221.5 2698.22   259.3 2675.47   292.5 2659.59   309.9 2647.23   321.9 2636.99
     330 2627.66   332.9 2626.17   354.1 2624.12   374.2 2626.15   382.2 2629.23
   401.6 2632.37   430.4 2631.39   462.5 2633.81   494.7 2649.34   550.9  2667.9
   649.4 2680.91   695.5  2692.8   719.6 2696.83   731.7 2700.41   763.8 2705.18
   783.9 2711.36   799.9 2719.14     820 2720.84   830.5 2729.14   875.4 2752.52
#Mann= 3 ,-1 , 0
       0      .1       0   332.9    .045       0   374.2      .1       0
Bank Sta=332.9,374.2
XS Rating Curve= 0 ,0
Exp/Cntr(USF)=0,0
Exp/Cntr=0.3,0.1

Type RM Length L Ch R = 1 ,6062    ,231.2,238.7,253.1
XS GIS Cut Line= 4
     2420920.226      696844.3552420550.16702421696857.209092264
2420371.64717235696996.6574339592420047.01663523696941.161478435
#Sta/Elev= 30
       0 2727.19   145.6 2694.93   245.6 2684.87   305.7  2675.1   329.7 2667.33
   370.3 2648.93     400 2639.56   416.7 2636.21   419.5 2633.91   425.2  2624.5
   430.9  2618.1   453.7 2615.71     464 2612.95   477.3 2615.79   487.9 2618.94
   510.7 2620.48   522.5 2623.95   535.5 2631.28   559.1 2648.97   601.8 2662.87
   626.1  2667.7   711.4 2675.64   727.3 2680.66   755.1 2685.35   796.4    2698
   804.7 2698.69     825 2709.66   845.3  2711.1   857.4 2718.42   926.2 2741.93
#Mann= 3 ,-1 , 0
       0      .1       0   453.7    .045       0   477.3      .1       0
Bank Sta=453.7,477.3
XS Rating Curve= 0 ,0
Exp/Cntr=0.3,0.1

Type RM Length L Ch R = 1 ,5823    ,476.8,487.4,491.4
XS GIS Cut Line= 3
2420899.89470677696826.8657710252420575.04363843696774.104255631
2420059.02625291696582.311645559
#Sta/Elev= 30
       0 2716.91    74.1 2697.09    93.3 2693.37   175.4  2684.3   265.9 2671.57
   296.6  2662.1     355 2635.86   367.8 2633.04   394.1 2630.76   427.6 2617.08
   440.7 2614.19   453.1 2609.39   470.2 2607.05   488.72608.809   508.7 2608.38
   515.4 2609.53     530 2618.91   576.9 2634.14   590.1 2636.67   618.1 2650.35
   632.4 2660.12   649.5  2661.5   661.6 2671.61   666.5 2674.23   786.1 2729.95
   811.6 2744.17   837.2 2756.32     855 2766.53   873.2 2781.17   879.6  2784.4
#Mann= 3 , 0 , 0
       0      .1       0   488.7    .045       0   515.4      .1       0
Bank Sta=488.7,515.4
XS Rating Curve= 0 ,0
Exp/Cntr=0.3,0.1

Type RM Length L Ch R = 1 ,5336    ,188.8,190.6,188.7
XS GIS Cut Line= 2
2420885.51029738696733.0498082552420429.27043275696082.960111408
#Sta/Elev= 30
       0 2689.07   109.3 2670.86   138.5 2664.52   168.8 2654.74     239 2624.39
   271.4 2608.08     291 2601.54   319.4 2589.94     328  2588.5     346 2589.42
   354.5 2586.86   364.3 2581.84   371.1  2581.5   398.5 2580.94   413.1 2579.04
   415.6 2581.59   422.9  2590.1   447.3 2602.37   466.9 2605.71   534.8 2611.03
   563.5 2620.03   575.8 2622.54   592.2 2630.41   608.6 2631.98   620.9 2639.18
   675.5 2664.51   735.9 2698.08   755.9 2707.08   784.5 2723.61   794.2 2727.68
#Mann= 3 ,-1 , 0
       0      .1       0   371.1    .045       0   415.6      .1       0
Bank Sta=371.1,415.6
XS Rating Curve= 0 ,0
Exp/Cntr=0.3,0.1

Type RM Length L Ch R = 1 ,5145    ,400.1,398.8,392.9
XS GIS Cut Line= 2
 2421027.5653028696639.173202921 2420577.0113028695943.760202921
#Sta/Elev= 30
       0 2680.72    18.2 2675.37    35.5 2672.27     157 2654.42   214.8 2641.29
   229.6 2636.17   240.9 2629.98   273.7 2602.78   295.8 2588.05   324.4 2578.94
   347.3 2575.11   385.5 2566.38   400.7  2564.6   417.3 2566.79   438.8 2567.84
   454.9 2579.21   471.9 2588.08     477 2589.53   498.3 2592.37   572.3 2595.88
     614 2601.04   629.5 2607.41   653.3 2622.67   670.9 2625.67   678.3 2633.22
   691.4 2642.12   712.3 2652.59   752.8 2677.99   786.8 2695.85   828.6 2720.86
#Mann= 3 ,-1 , 0
       0      .1       0   385.5    .045       0   417.3      .1       0
Bank Sta=385.5,417.3
XS Rating Curve= 0 ,0
Exp/Cntr=0.3,0.1

Type RM Length L Ch R = 1 ,4746    ,323.1,310.7,300.3
XS GIS Cut Line= 2
2421395.79283801696336.614476246     2420803.153      695746.308
#Sta/Elev= 30
       0 2660.22     120 2639.84   137.7  2635.1   154.7 2632.37   206.5  2620.7
     248  2608.7   276.3 2597.58   304.6 2582.47   332.9 2563.12   340.2 2559.36
   374.1 2552.81   395.1 2550.47   404.9 2546.26   410.5 2545.29   421.9 2543.14
   438.9 2543.61   444.5 2545.44   470.1 2548.56   485.6    2552   513.9 2565.45
   526.5 2568.57   597.6 2568.33   618.6 2570.17   673.3 2579.83   705.3 2587.18
   729.8 2594.42   756.3 2609.59   771.3 2610.92   790.3 2624.71   836.5 2647.93
#Mann= 3 ,-1 , 0
       0      .1       0   410.5    .045       0   444.5      .1       0
Bank Sta=410.5,444.5
XS Rating Curve= 0 ,0
Exp/Cntr=0.3,0.1

Type RM Length L Ch R = 1 ,4436    ,431.5,450,448.2
XS GIS Cut Line= 3
     2421694.215      695940.943     2421312.314      695834.697
     2420852.973        695683.1
#Sta/Elev= 30
       0 2652.24    17.5  2647.1    99.1 2637.26   190.4 2619.09   285.9 2603.76
   294.2 2600.16   332.6 2570.25   339.1 2563.74     352 2546.74   364.8  2534.9
   370.2 2531.36   377.3 2529.67   389.7 2529.47   414.9 2531.53   441.8 2535.13
   467.2 2531.47   482.3    2532   494.9 2535.32   510.7 2537.13   545.5 2545.52
   562.3 2551.36   591.8 2550.63   629.7 2553.99   723.7 2571.98   745.9 2580.81
   765.9 2593.78   780.7 2595.92   785.6 2597.86     806 2614.52   880.1  2658.5
#Mann= 3 ,-1 , 0
       0      .1       0   370.2    .045       0   414.9      .1       0
#XS Ineff= 2 , 0
                          444.44         2538.98
Permanent Ineff=
       F       F
Bank Sta=370.2,414.9
XS Rating Curve= 0 ,0
Exp/Cntr=0.3,0.1

Type RM Length L Ch R = 1 ,3986    ,610,620.3,618.9
XS GIS Cut Line= 3
     2421732.276      695662.878     2421288.809      695402.471
2420947.69175842695220.910708896
#Sta/Elev= 30
       0 2604.37    62.1 2585.74    94.6 2578.13   176.5  2563.5   233.7 2549.55
   289.4 2541.88     345 2539.29     359 2533.06     384  2514.5   391.4 2510.93
   419.3 2510.73   447.1 2513.31   465.6 2509.69   474.9 2509.26   497.6 2506.78
   527.3 2509.76   533.2  2511.3   552.9 2525.13     559  2528.2   565.8 2529.71
   583.5  2529.7   611.8 2539.03   670.7 2562.26   695.9 2575.04   725.5 2592.67
   778.7 2628.68   793.5 2640.17   843.7 2684.31   883.6 2715.64   900.7 2726.58
#Mann= 3 ,-1 , 0
       0      .1       0   474.9    .045       0   527.3      .1       0
#XS Ineff= 2 , 0
          441.99 2520.79
Permanent Ineff=
       F       F
Bank Sta=474.9,527.3
XS Rating Curve= 0 ,0
Exp/Cntr=0.3,0.1

Type RM Length L Ch R = 1 ,3365    ,124,129.7,133.1
XS GIS Cut Line= 2
2422090.13467076695236.6776168572421334.77700266694826.701954662
#Sta/Elev= 30
       0  2562.4    90.3 2548.43   163.1 2538.72   210.3  2534.1     290 2520.69
   299.7 2515.98   313.3 2505.02   354.3 2478.45   375.5 2472.19   397.9 2468.17
   404.4 2467.66   438.62468.758   449.9 2469.34   468.1 2473.72   481.7    2473
   504.5 2474.56   513.6 2477.92   545.4 2493.81   554.6 2492.36   568.2 2495.11
   624.3 2495.37   657.8 2506.45   673.5 2513.46     700 2529.72   717.7 2533.97
     732 2546.08     750  2558.6   791.5 2583.88   840.1 2617.06   859.4 2627.06
#Mann= 3 , 0 , 0
       0      .1       0   397.9    .045       0   438.6      .1       0
Bank Sta=397.9,438.6
XS Rating Curve= 0 ,0
Exp/Cntr=0.3,0.1

Type RM Length L Ch R = 1 ,3236    ,302.1,300,297.2
XS GIS Cut Line= 3
     2422110.561      695198.481     2421798.017      694933.643
     2421492.483      694661.034
#Sta/Elev= 30
       0 2553.18    67.9 2540.14   136.1  2532.2   269.2 2509.04   283.4 2504.37
   293.4 2499.15   303.8 2496.18   319.6 2488.86   339.7 2477.48     352 2468.75
   382.5  2454.3   389.2 2452.35   408.3 2450.81   431.8 2452.27   445.1  2463.5
   464.9 2470.43   489.1 2473.78   513.1 2473.78   544.2 2475.82   553.4 2478.01
     570 2485.08   615.1 2511.73   637.7 2528.62   671.4 2549.27   690.2 2563.19
   702.9 2565.22   705.7  2566.8   714.2 2575.36   726.2 2584.16   819.1 2640.76
#Mann= 3 ,-1 , 0
       0      .1       0   389.2    .045       0   431.8      .1       0
Bank Sta=389.2,431.8
XS Rating Curve= 0 ,0
Exp/Cntr=0.3,0.1

Type RM Length L Ch R = 1 ,2936    ,316.9,308.3,299.4
XS GIS Cut Line= 3
     2422345.951      694940.232     2422004.453      694718.639
     2421652.547      694483.666
#Sta/Elev= 30
       0 2539.11    46.7 2521.09    75.3 2508.15    89.7 2503.63     123 2503.12
   156.4 2497.25   194.1    2486   237.5 2480.06   257.8 2475.38   280.4 2467.67
   309.8 2449.47   318.4 2446.17   370.6  2443.7   386.6 2439.52   404.4 2437.25
   425.4 2439.45     438 2446.14   452.4  2459.5   493.1  2463.5   505.3 2473.06
   563.1 2504.58   638.9  2535.9   664.1 2549.14   697.7 2562.91   769.9 2598.87
   780.2 2602.66   793.9 2611.12   813.2 2615.35   822.8 2622.85   830.2  2626.4
#Mann= 3 ,-1 , 0
       0      .1       0   386.6    .045       0   425.4      .1       0
Bank Sta=386.6,425.4
XS Rating Curve= 0 ,0
Exp/Cntr=0.3,0.1

Type RM Length L Ch R = 1 ,2627    ,316.1,317.8,322.7
XS GIS Cut Line= 2
     2422568.948      694458.716 2421716.9966285694488.511716939
#Sta/Elev= 30
       0 2545.31    35.3 2534.08    70.2 2520.99   154.3 2481.37   218.3 2454.29
   238.3  2448.5   270.4 2444.58   313.2 2446.58   329.8 2445.34   338.1 2442.39
   354.4  2433.4   366.4 2424.09   378.4 2423.22   394.4 2422.66   408.4 2423.35
   430.5 2424.14   446.5 2429.27   466.5 2426.42   494.5 2431.44   526.5 2431.93
   574.6 2466.83   594.6 2468.91   606.6 2477.46   642.6 2496.27   690.6 2517.66
   702.6 2519.87   713.9 2524.23   733.2 2536.67   802.6 2566.11   852.5 2592.62
#Mann= 3 ,-1 , 0
       0      .1       0   378.4    .045       0   408.4      .1       0
#XS Ineff= 2 , 0
                          447.48         2431.34
Permanent Ineff=
       F       F
Bank Sta=378.4,408.4
XS Rating Curve= 0 ,0
Exp/Cntr=0.3,0.1

Type RM Length L Ch R = 1 ,2310    ,281.2,293.3,299.1
XS GIS Cut Line= 2
2422573.54206909694209.7308444512421674.33189657694159.569723645
#Sta/Elev= 30
       0 2545.83    50.9 2532.81     103 2513.24     131 2499.54   211.1 2445.93
   243.2 2431.96   267.2 2427.97   331.3 2425.03   363.4 2413.55   383.4 2418.23
   391.4 2418.49   407.3 2416.86   439.5 2408.22   459.5 2407.96   472.1 2410.54
   494.8 2406.23   523.6 2404.24   532.8  2405.7   555.7  2421.6   575.7 2439.03
   591.7 2447.87   611.7 2450.59   619.8 2456.63   653.4 2470.86   691.5 2491.99
     764 2527.59     776 2535.82     792 2540.39   810.3 2550.73   900.6 2591.74
#Mann= 3 ,-1 , 0
       0      .1       0   494.8    .045       0   532.8      .1       0
#XS Ineff= 2 , 0
          472.96 2412.89
Permanent Ineff=
       F       F
Bank Sta=494.8,532.8
XS Rating Curve= 0 ,0
Exp/Cntr=0.3,0.1

Type RM Length L Ch R = 1 ,2016    ,279,280.6,270
XS GIS Cut Line= 2
     2422587.968      694203.093     2421892.007      693733.966
#Sta/Elev= 30
       0 2548.81    78.7 2529.41   170.3 2498.53   237.8 2468.06   276.4 2444.81
   290.9 2438.53   322.4 2420.74   329.5 2418.09     344 2417.02     359 2412.45
     367 2408.49   377.7 2398.96     390  2392.1   401.9 2389.58   415.4 2387.42
   441.9 2389.09   458.4 2400.32   498.3 2409.73   565.9 2414.51     590    2418
   603.3 2422.35   618.9 2422.18   626.3 2424.29   658.7  2427.9   749.2 2456.53
   766.1 2460.46   778.1 2459.68   782.9 2461.01   816.7 2479.27   839.3 2485.55
#Mann= 3 ,-1 , 0
       0      .1       0   401.9    .045       0   441.9      .1       0
Bank Sta=401.9,441.9
XS Rating Curve= 0 ,0
Exp/Cntr=0.3,0.1

Type RM Length L Ch R = 1 ,1736    ,405.1,416.9,422.3
XS GIS Cut Line= 3
     2422725.866      693902.991     2422327.489      693722.901
     2421956.931      693559.294
#Sta/Elev= 30
       0  2517.6    69.3 2496.65   174.8 2457.44   205.4 2444.27   231.7 2429.94
   262.4 2417.97   293.1 2400.06   316.8 2390.21   330.4 2387.83   359.2 2388.74
   377.3 2382.46   394.1 2381.63   417.8 2376.39   429.2 2374.09   446.9 2374.36
   454.3 2376.69   474.2 2385.38   489.3 2395.69   503.6 2397.59   516.6 2403.67
     566  2406.2   608.5 2410.47   634.8 2416.88   647.9 2424.04   717.8 2455.01
   757.2 2477.97   779.1 2494.52   795.7 2499.89   803.6 2507.33   842.3 2531.01
#Mann= 3 ,-1 , 0
       0      .1       0   417.8    .045       0   454.3      .1       0
Bank Sta=417.8,454.3
XS Rating Curve= 0 ,0
Exp/Cntr=0.3,0.1

Type RM Length L Ch R = 1 ,1319    ,284.4,280.5,270.4
XS GIS Cut Line= 3
2422861.95946546693798.1091381772422627.10946546693462.093138178
2422375.94246546693138.749138177
#Sta/Elev= 30
       0 2518.88    76.4 2495.84   125.3 2478.66   213.8 2439.58   251.7 2420.13
   277.5 2405.35   354.7 2368.06     378 2361.79   404.1 2359.36   417.1 2359.54
   423.9 2357.28   435.3 2354.97   459.6 2357.27   480.9 2360.26   489.5 2364.54
     498 2366.78   514.9 2367.48   534.4 2365.72   540.8  2367.5   555.8 2375.87
   580.1 2384.71   619.2 2404.35   641.9 2417.94   652.1 2430.66   657.1 2434.79
   667.3  2438.3   731.8 2471.16   782.2  2488.7   808.7 2500.78   819.4 2504.09
#Mann= 3 ,-1 , 0
       0      .1       0   423.9    .045       0   459.6      .1       0
Bank Sta=423.9,459.6
XS Rating Curve= 0 ,0
Exp/Cntr=0.3,0.1

Type RM Length L Ch R = 1 ,1038    ,279.4,277.8,271.9
XS GIS Cut Line= 2
2423185.68796565693452.4000860632422426.94777576693062.583758785
#Sta/Elev= 30
       0 2523.13    29.6 2513.55    68.7  2498.2    99.6 2489.43   124.7 2478.24
   201.2  2448.5   228.2 2436.22     241  2423.8   255.1 2414.14   300.4 2387.61
   318.2 2379.42   359.8 2349.29   376.6 2344.38   392.5 2345.98   403.5 2342.44
   412.5  2341.1   428.1 2341.47   434.1 2343.35   448.9 2353.52   493.5 2349.34
   508.3 2351.58   526.2 2351.19   561.8 2359.61   574.4 2366.22   587.9  2368.7
   600.4 2375.07   623.9 2381.83   664.4 2396.91   781.3  2448.7     853 2483.12
#Mann= 3 ,-1 , 0
       0      .1       0   403.5    .045       0   434.1      .1       0
Bank Sta=403.5,434.1
XS Rating Curve= 0 ,0
Exp/Cntr=0.3,0.1

Type RM Length L Ch R = 1 ,761     ,103.4,99.6,100.3
XS GIS Cut Line= 2
2423270.15057955693091.3379144762422483.76964779692922.363499387
#Sta/Elev= 30
       0 2471.54    40.3 2466.03    64.9 2459.22   101.7 2447.03   142.6 2429.23
     159 2420.24   171.2 2407.84   183.5 2399.32   228.9 2372.84   240.8 2362.92
   249.1 2350.72   261.2 2344.43   289.5 2342.43   326.9 2345.68   383.8 2334.67
   392.2 2331.11   412.6 2330.45   424.9 2333.83     429 2334.86   449.4 2332.24
   486.3 2334.34   498.3 2341.53   519.7 2361.66   527.2 2366.91   552.2 2367.46
   576.3 2370.96   592.6 2380.69   629.5 2390.43   727.6 2427.73   804.3 2451.99
#Mann= 3 , 0 , 0
       0      .1       0   383.8    .045       0   424.9      .1       0
Bank Sta=383.8,424.9
XS Rating Curve= 0 ,0
Exp/Cntr(USF)=0,0
Exp/Cntr=0.3,0.1

Type RM Length L Ch R = 1 ,661     ,290.4,288.8,290.4
XS GIS Cut Line= 3
2423298.08161382692998.2203170942422868.61461382692907.368317093
2422475.69361382692812.129317094
#Sta/Elev= 30
       0 2457.31      32 2449.16    93.4 2429.59   146.5 2408.28   248.6  2355.7
     279 2334.86     306 2333.22   326.4 2336.39   350.9 2335.29   373.5 2338.23
     400 2338.24   408.2 2336.11   427.5 2325.49     445 2322.63   457.4 2325.32
   482.1  2326.6   490.3 2329.22     515 2344.94   531.4  2358.1     552 2361.43
   576.7 2371.13   589.1 2373.14   609.6 2382.49   642.6 2389.26   654.9 2394.41
   745.5 2422.86   774.3 2439.94   786.6 2443.31   799.4 2451.12   843.3 2472.28
#Mann= 3 ,-1 , 0
       0      .1       0   427.5    .045       0   457.4      .1       0
Bank Sta=427.5,457.4
XS Rating Curve= 0 ,0
Exp/Cntr=0.3,0.1

Type RM Length L Ch R = 1 ,372     ,209.9,216.9,219.9
XS GIS Cut Line= 2
2423392.45117807692753.0985120382422567.21724376692554.482887168
#Sta/Elev= 30
       0 2414.19   104.6 2370.78     151 2349.02   178.7  2339.5   252.7 2338.04
     261    2336   285.6 2320.24   293.9    2317   306.2  2316.5   318.5 2318.73
   339.1 2319.71   359.7 2313.67   388.5 2309.85   409.1 2308.54   419.7 2309.95
   446.1 2309.18   462.5 2319.18     479 2331.62   491.3 2333.62   511.9 2343.54
   528.4 2356.28     557  2372.3   569.5 2378.08   626.7 2398.56     660 2416.62
   676.4 2427.59   689.7  2431.6   709.1 2441.19   738.2 2452.88   848.8 2493.88
#Mann= 3 ,-1 , 0
       0      .1       0   388.5    .045       0   419.7      .1       0
Bank Sta=388.5,419.7
XS Rating Curve= 0 ,0
Exp/Cntr(USF)=0,0
Exp/Cntr=0.3,0.1

Type RM Length L Ch R = 1 ,155     ,132.9,155.1,132.9
XS GIS Cut Line= 4
2423346.57382945692706.9075409552423225.82101672692561.760220607
2422987.97456741692415.3931748782422719.63498358 692406.85509721
#Sta/Elev= 30
       0 2383.83    28.3 2371.17    73.7 2346.37    93.7 2338.92   116.3 2334.23
     176 2330.91   230.9 2327.49   239.7 2323.59   258.2 2310.31   271.6 2302.07
   278.2 2300.32   291.1 2300.18   298.32298.873   306.5 2298.07   331.1 2299.31
   342.7  2301.8   356.8 2309.35   361.5 2310.81   375.6 2312.41   414.1 2312.97
   446.1 2323.29   457.7 2329.22   489.3 2352.04   501.3 2369.09   509.3 2376.61
   545.4 2396.82   582.2 2420.91   617.6 2435.65   657.4 2448.41   736.6 2468.78
#Mann= 4 ,-1 , 0
       0     .06       0     176      .1       0   298.3    .045       0
   331.1      .1       0
Bank Sta=298.3,331.1
XS Rating Curve= 0 ,0
Exp/Cntr(USF)=0,0
Exp/Cntr=0.3,0.1

Type RM Length L Ch R = 1 ,0       ,,,
XS GIS Cut Line= 4
2423527.68982637692222.4890393612423290.35876885692360.781206399
2423197.69999999692365.1560000032422771.26154664692377.274261966
#Sta/Elev= 30
       0 2400.57    24.2 2384.55    79.8 2359.33   121.5 2336.07   150.2 2323.13
   170.6    2310   190.9 2306.28   226.2 2307.22   246.5 2310.55     263 2306.11
   274.7 2299.52   302.3 2295.55   310.3 2297.68   341.3 2295.67   356.1 2290.58
   366.4 2288.59   386.4 2290.53   398.4 2293.25   414.4 2306.62   426.4 2308.56
   438.4 2311.02   518.5 2314.23   538.5 2317.66   562.5  2332.7   610.5 2372.67
   652.2 2395.18   674.5  2409.7   702.7  2424.2   742.6 2440.55794.0556 2453.37
#Mann= 5 ,-1 , 0
       0      .1       0   226.2     .06       0   356.1    .045       0
   386.4     .06       0   426.4      .1       0
Bank Sta=356.1,386.4
XS Rating Curve= 0 ,0
Exp/Cntr(USF)=0,0
Exp/Cntr=0.3,0.1
LCMann Table=0

Chan Stop Cuts=-1
Use User Specified Reach Order=0
Composite Channel Slope=5
